HEC-RAS study 17465_ras.prj: 17465

--- 17465_ras.g01 (geometry) --- (continued)

Type RM Length L Ch R = 1 ,35138.73,149.015600,149.015600,149.015600
XS GIS Cut Line= 6
788328.738962064784233.381241247788518.426801756784307.716157421
788987.102737025784498.048179368789366.188346289784659.598014198
789901.978955074784896.183059467790044.444990796784956.472354599
#Sta/Elev= 30
8928.375502.1214 8945.84501.01999021.023472.20059069.849464.89859149.996423.6169
9279.514382.55349430.618376.05549473.791360.62189523.548359.19149570.929335.9753
9592.515334.89939624.895325.83629668.297327.99739700.923324.75419733.549332.7858
9787.926335.00239842.303343.3714 9874.93329.83619972.808326.88669994.559321.6075
10027.07327.267910063.41325.047810103.39342.576210114.32343.664810201.78333.9626
10310.97342.390110507.86396.902910573.45399.543210671.59447.763910790.43450.9766
#Mann= 3 , 0 , 0
8928.375   0.075       08928.375   0.075       010790.43   0.075       0
#XS Ineff= 2 , 0
       09843.268        10117.62       0
Bank Sta=8928.375,10790.43
Exp/Cntr=0.3,0.1

Type RM Length L Ch R = 1 ,34989.72,149.015700,149.015700,149.015700
XS GIS Cut Line= 6
788244.623698686 784334.19618047788601.192222105784476.046746684
788871.898177652 784591.29375564789347.269876951784812.814933617
789670.875213098784970.789368179790080.096666225785149.741963497
#Sta/Elev= 30
8877.345488.75298960.878476.35319028.398457.55359060.688439.56089103.742 433.981
9157.559409.66329179.086391.15389308.564381.92569341.073363.18039384.417354.9933
9439.582358.46159515.061 343.0559735.547324.96739780.249326.4405  9802.6339.5244
9824.951340.87849869.653326.328710001.55321.6392 10055.8326.951210099.69343.8919
10166.45335.437810233.22334.787710333.37347.4028 10532.6361.1113 10576.6381.4133
10609.43388.241910631.28399.362810653.13401.048110751.12442.730710886.75 437.156
#Mann= 3 , 0 , 0
8877.345   0.075       08877.345   0.075       010886.75   0.075       0
#XS Ineff= 2 , 0
       09834.164        10103.11       0
Bank Sta=8877.345,10886.75
Exp/Cntr=0.3,0.1

Type RM Length L Ch R = 1 , 34840.7,149.015600,149.015600,149.015600
XS GIS Cut Line= 6
788191.758560655784423.406100874788909.655453054784724.087712832
789072.644154088784813.476304519789408.217347624785054.933554585
789740.743199498785217.445484823790110.108158841785368.642274575
#Sta/Elev= 30
8894.605489.32179037.795437.99769144.974412.64399177.234397.7628 9285.25388.3888
9328.533364.32479350.174364.69359393.496378.30579491.699373.84649590.661378.4483
 9634.87350.05749668.027337.59869724.262335.7711 9769.33325.01519827.103323.2248
9838.685327.61629886.115323.09949910.263328.3631    9999320.128510092.27326.2375
10138.94 343.23610269.91331.4906 10337.4334.264710402.94 346.52710450.09335.4966
10527.26335.391610757.08365.544710876.35405.051510919.33428.597911042.99 426.918
#Mann= 3 , 0 , 0
8894.605  0.0698       08894.605  0.0698       011042.99  0.0698       0
#XS Ineff= 2 , 0
       0 9869.12        10143.32       0
Bank Sta=8894.605,11042.99
Exp/Cntr=0.3,0.1

Type RM Length L Ch R = 1 ,34691.69,149.015600,149.015600,149.015600
XS GIS Cut Line= 6
788203.383393364784626.501763673788690.938991801784822.580225501
788925.718755789 784932.54912529789459.318408183785208.780409826
  789805.5110956785362.160274729790081.865278244785468.393725199
#Sta/Elev= 30
9014.424448.07829101.687 422.1669176.759410.73399316.651378.65679588.374369.0798
9720.638369.27279742.876372.34389753.995369.5032 9799.27341.95479854.643339.2346
9899.588322.3284 9955.77324.801810002.05320.677510102.31325.0775 10152.1341.3202
10204.36334.8203 10272.4337.332710305.94332.526110328.29339.225410346.89 340.134
10438.87331.019910516.56334.675310658.75356.681210756.57357.258210810.58369.9963
10875.12374.785810918.15384.917610971.74402.9602 11003.8420.301811074.95422.8137
#Mann= 3 , 0 , 0
9014.424  0.0774       09014.424  0.0774       011074.95  0.0774       0
#XS Ineff= 2 , 0
       09882.504         10163.2       0
Bank Sta=9014.424,11074.95
Exp/Cntr=0.3,0.1

Type RM Length L Ch R = 1 ,34542.67,149.015700,149.015700,149.015700
XS GIS Cut Line= 6
788178.215671743784817.166321462788452.905547756 784920.67052989
788980.764981984785137.688158429789111.256791301785183.621095081
789758.604945123785461.101502559790053.296331951785569.296812108
#Sta/Elev= 30
9069.898 442.1589119.713431.47349194.376423.91639258.619424.8987 9333.57411.5805
9354.984405.09989387.253379.7411  9408.8372.95459635.298370.21559722.008360.2784
9787.041342.5635 9884.59340.86639917.106326.77439970.725319.370110023.13318.9773
 10065.9324.974710109.49321.857810164.13 341.647 10274.3340.616810382.71 330.988
10491.75330.780910567.89346.127410643.57342.679610708.33351.933310773.09351.2318
10869.41368.049110922.91381.848910976.08402.558611029.11414.348411090.92420.1316
#Mann= 3 , 0 , 0
9069.898  0.0792       09069.898  0.0792       011090.92  0.0792       0
#XS Ineff= 2 , 0
       0                10166.33       0
Bank Sta=9069.898,11090.92
Exp/Cntr=0.3,0.1

Type RM Length L Ch R = 1 ,34393.65,149.015600,149.015600,149.015600
XS GIS Cut Line= 6
788155.353249358784990.366491086788932.476020309785275.970467309
789240.079590896785391.358677476789645.017415835785548.938651458
789864.989692982785628.928254743790021.689652239785680.928914924
#Sta/Elev= 30
9117.141432.38089350.793431.79779361.454429.88379393.435398.19889436.078378.7557
9702.592359.20719740.295351.82869777.216336.4245  9862.5337.28039883.821344.4725
9926.464324.38679990.698319.6363   10119323.032510161.63340.915910225.59327.9707
10257.56326.963910393.98330.039610461.34341.246710525.72 334.63310622.29336.9287
10686.68349.507510740.06340.020810825.18344.479710867.75355.356110889.03368.4515
10910.31373.351611005.45413.377811037.06412.160211068.67426.091611107.32427.5624
#Mann= 3 , 0 , 0
9117.141   0.085       09117.141   0.085       011107.32   0.085       0
#XS Ineff= 2 , 0
       0                10171.78       0
Bank Sta=9117.141,11107.32
Exp/Cntr=0.3,0.1

Type RM Length L Ch R = 1 ,34244.64,149.015600,149.015600,149.015600
XS GIS Cut Line= 6
788131.758569935785169.114062522788755.049054136785385.055082797
789041.140299622785464.780297048789145.467276173785497.285341057
789685.118625576785689.980524577789991.555063722785787.361716923
#Sta/Elev= 30
9139.858 463.6389259.384460.38269291.188431.92539333.594427.66349397.203402.5776
9471.414 380.1279535.023372.58179556.226364.70219641.037350.95229683.331336.8732
9746.672331.40159872.606335.1882 9920.06316.226210007.46313.3925 10090.2316.6486
10132.02336.667110258.24328.448410332.32338.125310410.01329.699610481.13327.4405
 10616.6341.785710704.33334.090410789.27338.922410831.43349.5855 10905.2382.0105
10926.27386.315110947.32398.102811041.59 430.85611072.81435.333111100.44433.9867
#Mann= 3 , 0 , 0
9139.858   0.075       09139.858   0.075       011100.44   0.075       0
#XS Ineff= 2 , 0
       0                10160.28       0
Bank Sta=9139.858,11100.44
Exp/Cntr=0.3,0.1

Type RM Length L Ch R = 1 ,34095.62,149.015700,149.015700,149.015700
XS GIS Cut Line= 6
788113.037219457785310.942475271788388.026500904785403.347355259
789403.815830111785756.490579197789637.940341347785833.838002312
789794.337880813785880.993503076 789952.85672881785924.040942363
#Sta/Elev= 30
9166.774462.69549295.432460.42019337.632430.06139348.181426.49559390.381425.0372
9548.943371.63179580.701369.66049665.388353.34139728.904333.32859845.349329.7434
9877.107326.30129908.865311.41529930.036307.739410010.49306.075810110.03311.3717
10141.79326.887610215.91328.204210332.38320.176610427.67324.223110527.76338.2594
10670.46328.475810786.24 336.78710880.24 375.63310901.13380.151310922.02391.8271
10942.91396.383610963.63410.011110984.36 412.924 11025.8 435.00411106.48437.2194
#Mann= 3 , 0 , 0
9166.774   0.075       09166.774   0.075       011106.48   0.075       0
#XS Ineff= 2 , 0
       0                10159.66       0
Bank Sta=9166.774,11106.48
Exp/Cntr=0.3,0.1

Type RM Length L Ch R = 1 ,33946.61,149.015600,149.015600,149.015600
XS GIS Cut Line= 6
788094.480104076785451.526682742788611.804582037785627.187061389
789029.304866312785792.431021781789308.357353702785893.381661283
789665.183803261786000.685143325789914.165382553786060.695484465
#Sta/Elev= 30
9191.801459.09719265.819457.62039307.803426.97479444.631424.8267 9455.19419.7767
9486.866417.3216  9529.1391.92789560.788379.6204 9582.06367.40459645.878354.7846
9688.422352.12339738.205331.7472  9881.4327.35759924.403310.7192 9999.66306.0992
10074.98  311.8810107.26310.0412 10150.3327.560310203.99322.337610363.98319.1781
10416.92328.783610522.46323.517910721.22332.867210794.04361.143210825.25368.9288
10877.08405.041310915.29 412.79910969.89433.994410997.24438.011311112.79438.6388
#Mann= 3 , 0 , 0
9191.801   0.075       09191.801   0.075       011112.79   0.075       0
#XS Ineff= 2 , 0
       0                10162.02       0
Bank Sta=9191.801,11112.79
Exp/Cntr=0.3,0.1

Type RM Length L Ch R = 1 ,33797.59,149.015600,149.015600,149.015600
XS GIS Cut Line= 6
788244.633251103785642.888265048788660.553259882785791.613456925
788855.643060111785892.652390236 789087.50625859785988.170645793
789386.196117191786081.458944173789885.815846433786194.711500688
#Sta/Elev= 30
9418.285424.91099471.217426.57159481.726424.07199513.253397.79549534.271396.4183
9565.799 375.7719597.462362.57219676.754352.6527 9714.25 332.4889757.084329.4728
9909.431328.09399954.007309.10819999.647304.321310090.24311.620910145.15310.2198
10178.09325.413210189.03327.475610296.05318.551210412.49 314.602 10652.9328.6149
10683.86338.241810704.51340.249310766.44373.010310797.41 377.047 10838.7399.9209
10869.55403.118810910.49428.359310920.72430.681410941.19434.914111156.27437.0032
#Mann= 3 , 0 , 0
9418.285   0.075       09418.285   0.075       011156.27   0.075       0
#XS Ineff= 2 , 0
       0                10195.76       0
Bank Sta=9418.285,11156.27
Exp/Cntr=0.3,0.1

Type RM Length L Ch R = 1 ,33648.58,149.015600,149.015600,149.015600
XS GIS Cut Line= 6
 788196.81280981785827.793971378788426.599306144785895.845151139
789072.706457874786102.542511725789285.815759389786163.045176389
789633.725795089 786241.91810382789868.107096619786281.484374787
#Sta/Elev= 30
9445.853394.9044 9516.77371.35099527.212372.3776  9543.6365.66959600.305353.6972
9642.072335.58029662.956 330.548 9925.15328.71879977.611306.75249998.595302.5523
10030.03 307.50310092.96305.850710156.04308.756310198.09327.645310261.16320.3989
10376.69316.019610397.54 312.468 10470.5 312.51910501.67318.825710553.49318.0915
10605.16322.068110687.49337.460410738.94359.170610769.81377.259810820.95398.2643
10923.08 400.86710953.65418.622710973.95422.977510994.25433.834411179.92434.0128
#Mann= 3 , 0 , 0
9445.853   0.075       09445.853   0.075       011179.92   0.075       0
#XS Ineff= 2 , 0
       0                10212.18       0
Bank Sta=9445.853,11179.92
Exp/Cntr=0.3,0.1

Type RM Length L Ch R = 1 ,33499.56,149.015700,149.015700,149.015700
XS GIS Cut Line= 6
788152.788083943785998.022911397789042.950080668786226.377319009
789258.504263125786277.523798688789448.041128039786316.181352433
789609.066194923786343.643916358789848.936129224786375.422115036
#Sta/Elev= 30
9444.878366.58529508.912356.2216 9539.79 346.9449591.343346.9624 9653.29 330.417
9921.726327.2959 9983.86304.687510004.58302.947910056.37304.961510097.73310.6524
10149.32 306.85810190.59325.370110200.91326.669410273.14317.775410386.55318.4795
10427.66 312.65210581.82315.195310612.46326.725510653.29330.541410683.91344.4721
10714.52350.877610755.35375.828810775.76382.903710796.07396.8477 10948.2398.7085
10978.48415.334810988.58413.991511018.86432.441611150.05433.582311184.19430.3512
#Mann= 3 , 0 , 0
9444.878   0.075       09444.878   0.075       011184.19   0.075       0
#XS Ineff= 2 , 0
       0                10206.99       0
Bank Sta=9444.878,11184.19
Exp/Cntr=0.3,0.1

Type RM Length L Ch R = 1 ,33350.54,149.015600,149.015600,149.015600
XS GIS Cut Line= 6
788108.278424612786170.126927478 788507.72304571786254.183121391
788771.806913576786299.870995958789231.794880787786390.319371472
 789499.75967757786432.159798526789830.556612449786465.481747242
#Sta/Elev= 30
9440.405342.52679508.588345.02339529.026342.26269549.464334.30559641.435334.0548
9672.092328.13489917.042326.66019957.654309.2096 10008.3302.509410059.01304.7066
10079.29 308.89810140.27306.299310191.26326.181610252.45320.854610395.22317.0459
10415.61312.456110558.15313.040510608.96332.773910649.53333.466810659.67341.0318
10673.33343.490910791.21394.736610851.84397.716410972.66395.410810982.72397.0433
11002.86411.355511012.92412.316511043.11 428.77311133.48430.351311189.17426.6504
#Mann= 3 , 0 , 0
9440.405  0.0562       09440.405  0.0562       011189.17  0.0562       0
#XS Ineff= 2 , 0
       0                10204.03       0
Bank Sta=9440.405,11189.17
Exp/Cntr=0.3,0.1

Type RM Length L Ch R = 1 ,33201.53,276.902800,276.902800,276.902800
XS GIS Cut Line= 6
788067.691119802786327.064506075788562.718686746786416.421235828
789212.771016973786519.468105371  789567.7824758786554.585960837
789765.162629021786564.988193042790135.557886762786570.582353302
#Sta/Elev= 30
9424.206337.58889451.956331.40969594.218332.12279899.067325.24339929.543310.8991
9959.918304.444210010.55301.915210051.09308.297710122.02308.875210172.69325.1612
10253.77318.077310375.38319.375910405.76312.874910476.51318.823910537.14334.7549
10627.92 340.08410668.18358.310310728.57376.847410758.76391.930910824.23399.2655
10969.47395.864910989.49399.138711009.52 413.17811019.54414.092111029.55419.9667
11239.73 421.19411269.74424.752811379.77474.454211399.77 487.14311510.33489.2351
#Mann= 3 , 0 , 0
9424.206  0.0548       09424.206  0.0548       011510.33  0.0548       0
#XS Ineff= 2 , 0
       0                10194.27       0
Bank Sta=9424.206,11510.33
Exp/Cntr=0.3,0.1

Type RM Length L Ch R = 1 ,32924.63,214.609300,214.609300,214.609300
XS GIS Cut Line= 6
788048.633629841786613.597540542788884.287937544786747.323530896
789114.733243118786767.777705645 789361.20075729786774.124535608
789524.542275821786772.271666669790079.125985146786622.532916442
#Sta/Elev= 30
9455.976323.67339533.048328.18399826.746327.59229877.512322.88829918.126304.5448
10009.49302.019910050.06306.085510090.63305.612510141.33325.931110232.36327.0901
10303.07354.624910513.95359.6783   10534365.330510564.03361.702410624.08365.3139
10634.08369.297810654.09371.1727 10694.1393.184311006.28394.6453   11027402.6361
11109.86407.016711130.58415.594811213.44413.467711296.31419.026811327.38428.1018
11358.46432.054411379.17 437.89311451.68471.1431 11472.4484.6088 11518.1 487.502
#Mann= 3 , 0 , 0
9455.976  0.0638       09455.976  0.0638       0 11518.1  0.0638       0
#XS Ineff= 2 , 0
       0                10183.61       0
Bank Sta=9455.976,11518.1
Exp/Cntr=0.3,0.1

Type RM Length L Ch R = 3 ,32820.61,,,
BEGIN DESCRIPTION:
END DESCRIPTION:
Bridge Culvert--1,0,-1,-1, 0
Deck Dist Width WeirC Skew NumUp NumDn MinLoCord MaxHiCord MaxSubmerge Is_Ogee
79.804650,55.000000,2.6,0, 60, 60, , , 0.95, 0, 0,0,,
 9224.50 9232.87 9252.98 9263.04 9293.22 9323.40 9333.46 9363.63 9373.69 9383.75
 9393.81 9403.87 9444.10 9464.22 9484.34 9494.40 9504.46 9544.69 9615.10 9645.28
 9685.52 9725.75 9835.83 9835.8310150.8310150.8310155.4210160.5010190.8910201.02
10211.1510241.5410251.6710261.8010322.5910535.3510565.7410575.8710646.7910687.32
10747.8210757.8310787.8410837.8710877.8911107.3611221.6011252.7611283.9211304.69
11325.4611335.8511367.0011377.3911387.7711398.1611408.5511418.9311429.3211444.22
  358.20  357.94  355.42  352.45  335.14  320.50  318.47  320.25  318.01  319.35
  323.16  325.04  325.73  326.81  329.01  326.64  326.05  326.32  329.23  331.09
  332.10  334.11  336.58  336.58  339.00  339.00  339.03  340.51  341.22  335.10
  326.08  325.42  337.29  344.29  348.14  365.27  367.20  368.86  373.97  377.83
  382.70  382.98  385.85  388.66  391.77  404.05  408.76  411.54  413.00  413.07
  414.14  415.45  415.64  416.62  424.12  436.86  439.78  441.08  442.02  441.98
 -641.80 -642.06 -644.58 -647.55 -664.86 -679.50 -681.53 -679.75 -681.99 -680.65
 -676.84 -674.96 -674.27 -673.19 -670.99 -673.36 -673.95 -673.68 -670.77 -668.91
 -667.90 -665.89 -663.42  334.08  336.50 -661.00 -660.97 -659.49 -658.78 -664.90
 -673.92 -674.58 -662.71 -655.71 -651.86 -634.73 -632.80 -631.14 -626.03 -622.17
 -617.30 -617.02 -614.15 -611.34 -608.23 -595.95 -591.24 -588.46 -587.00 -586.93
 -585.86 -584.55 -584.36 -583.38 -575.88 -563.14 -560.22 -558.92 -557.98 -558.02
 9224.50 9232.87 9252.98 9263.04 9293.22 9323.40 9333.46 9363.63 9373.69 9383.75
 9393.81 9403.87 9423.98 9444.10 9464.22 9484.34 9494.40 9504.46 9534.63 9725.75
 9844.38 9844.3810155.4210159.3810159.3810190.8910201.0210211.1510241.5410251.67
10261.8010322.5910535.3510565.7410575.8710646.7910687.3210747.8210757.8310787.84
10837.8710877.8911107.3611128.1311200.8311221.6011252.7611283.9211304.6911325.46
11335.8511367.0011377.3911386.0211387.7711398.1611408.5511418.9311429.3211444.22
  358.20  357.94  355.42  352.45  335.14  320.50  318.47  320.25  318.01  319.35
  323.16  325.04  324.97  325.73  326.81  329.01  326.64  326.05  326.11  334.11
  336.50  336.50  339.03  340.18  340.18  341.22  335.10  326.08  325.42  337.29
  344.29  348.14  365.27  367.20  368.86  373.97  377.83  382.70  382.98  385.85
  388.66  391.77  404.05  404.48  408.24  408.76  411.54  413.00  413.07  414.14
  415.45  415.64  416.62  422.46  424.12  436.86  439.78  441.08  442.02  441.98
 -641.80 -642.06 -644.58 -647.55 -664.86 -679.50 -681.53 -679.75 -681.99 -680.65
 -676.84 -674.96 -675.03 -674.27 -673.19 -670.99 -673.36 -673.95 -673.89 -665.89
 -663.50  334.00  336.53  337.68 -659.82 -658.78 -664.90 -673.92 -674.58 -662.71
 -655.71 -651.86 -634.73 -632.80 -631.14 -626.03 -622.17 -617.30 -617.02 -614.15
 -611.34 -608.23 -595.95 -595.52 -591.76 -591.24 -588.46 -587.00 -586.93 -585.86
 -584.55 -584.36 -583.38 -577.54 -575.88 -563.14 -560.22 -558.92 -557.98 -558.02
Pier Skew, UpSta & Num, DnSta & Num=  ,9911.58, 2 ,9920.13, 2 , 0 , 0 , 0 ,,
   12.00   12.00
 -662.95  337.05
   12.00   12.00
 -662.88  337.12
Pier Skew, UpSta & Num, DnSta & Num=  ,9993.33, 2 ,10001.88, 2 , 0 , 0 , 0 ,,
   12.00   12.00
 -662.29  337.71
   12.00   12.00
 -662.22  337.78
Pier Skew, UpSta & Num, DnSta & Num=  ,10075.08, 2 ,10083.63, 2 , 0 , 0 , 0 ,,
   12.00   12.00
 -661.62  338.38
   12.00   12.00
 -661.55  338.45
BR Coef=-1 , 0 , 0 ,, 0 ,,,0.8,0,1,0,
WSPro=,,,, 1 ,,,, 0 ,,,, 0 ,,,,-1 ,-1 ,-1 , 0 , 0 , 0 , 0 , 0
BC Design=,, 0 ,, 0 ,,,,,,

Type RM Length L Ch R = 1 ,32710.02,462.629700,462.629700,462.629700
XS GIS Cut Line= 6
788061.563934933786849.745744176788343.059864253786875.012174577
788751.078529716786941.703704581789067.841262966787021.838472009
789345.619040728 787026.17874977790187.632929623786809.164860889
#Sta/Elev= 30
9510.958 323.3719715.043321.36899825.945317.07689876.654 318.8579917.374299.3103
9927.553296.806110029.29295.805410100.38 296.45210150.78320.153410160.85322.8804
10231.92326.1485 10355.7340.898910631.16349.267110651.16 359.90910701.17380.3053
10751.17387.395711069.33391.143211079.66 388.03911100.31392.704911131.29403.9133
11162.27405.499111193.25410.572311255.21409.710111472.08 417.05211492.73422.6019
11523.71439.595811565.02446.646711585.67454.965311657.95470.105611681.33467.4079
#Mann= 3 , 0 , 0
9510.958  0.0861       09510.958  0.0861       011681.33  0.0861       0
#XS Ineff= 2 , 0
       0                10195.96       0
Bank Sta=9510.958,11681.33
Exp/Cntr=0.3,0.1

Type RM Length L Ch R = 1 ,32247.39,248.843600,248.843600,248.843600
XS GIS Cut Line= 6
788091.547716097787397.344274128788413.950419247787405.183924809
788640.370210767787334.030646205 789139.64774695787155.798733503
789485.610890269787068.712090686789877.187169552786989.638083607
#Sta/Elev= 30
9495.062320.94159558.533316.29579668.566319.6415 9881.92317.48119944.991 292.979
9965.838291.57659986.685286.217710017.98286.424410028.43292.489410051.58295.2619
10133.96 295.31810145.92298.300310178.18314.848510199.68315.076710253.44332.6009
10328.33333.533110360.16338.1773 10507.5338.880210528.37348.693710653.12349.4895
10673.84360.017710684.21 361.03510746.11387.285610848.97387.518510910.69383.9851
10951.78386.576911105.14384.725811115.36387.053511156.21406.744311341.68417.2712
#Mann= 3 , 0 , 0
9495.062   0.075       09495.062   0.075       011341.68   0.075       0
#XS Ineff= 2 , 0
       09851.608        10208.45       0
Bank Sta=9495.062,11341.68
Exp/Cntr=0.3,0.1

Type RM Length L Ch R = 1 ,31998.54,248.843500,248.843500,248.843500
XS GIS Cut Line= 6
787958.290364902787882.712135061788351.255437109787739.264133902
789048.631580395787363.701898577789217.927463852787288.601645411
789646.769374827787149.969481574790112.138547072787039.869512656
#Sta/Elev= 30
 9186.59329.06579351.343326.00349372.643316.20589400.459314.79979488.563314.4874
9539.116320.48969642.593319.38979675.851312.21039732.127290.80439847.184287.6006
9888.448 296.5259939.733290.79439961.842293.75639983.229285.922710003.69285.4724
10057.24294.5232 10105.6291.574510160.15313.114410233.36 318.986 10440.3323.8517
10495.36337.294810592.88  338.72 10656.9 354.62210699.57372.9133 10752.3377.0417
10909.53376.302411055.05380.865211075.68384.608711137.58408.805611514.52424.8707
#Mann= 3 , 0 , 0
 9186.59  0.0761       0 9186.59  0.0761       011514.52  0.0761       0
#XS Ineff= 2 , 0
       09840.281        10188.63       0
Bank Sta=9186.59,11514.52
Exp/Cntr=0.3,0.1

Type RM Length L Ch R = 1 , 31749.7,248.843600,248.843600,248.843600
XS GIS Cut Line= 6
788013.980208162788150.719505779788506.636553153787953.544510933
 789046.60738638 787624.53442289789418.595576639787435.565853175
789696.890448626787328.158152479790214.842702178787171.152215277
#Sta/Elev= 30
9062.599323.54549276.061323.01879351.453312.98099448.648 317.7859492.412313.5069
9797.598314.67749816.955311.98939856.054297.891810001.49283.374810011.27283.5783
10035.09292.4566   10047290.603410106.55312.812810165.54316.489510235.97 311.717
10418.63316.739810584.92348.5701 10606.9358.846810639.88362.192510801.65364.5702
10854.93370.041410982.31369.210111066.55400.124211111.96409.808211150.67409.1098
 11202.8416.274911223.66 413.49511338.34418.2112 11390.4415.524411483.52418.0586
#Mann= 3 , 0 , 0
9062.599   0.075       09062.599   0.075       011483.52   0.075       0
#XS Ineff= 2 , 0
       09787.977        10124.05       0
Bank Sta=9062.599,11483.52
Exp/Cntr=0.3,0.1

Type RM Length L Ch R = 1 ,31500.86,248.843600,248.843600,248.843600
XS GIS Cut Line= 6
788053.163552413788339.289350007788536.606765323788154.382206117
789092.863279042787915.350770281789823.310718439787586.028723532
790113.407200536787472.463872874790377.325993743787378.848248855
#Sta/Elev= 30
9017.764320.44339318.052320.41289344.708313.4878 9371.69312.5817 9817.69311.2311
9828.613309.85379861.384295.13979871.813293.20459934.452293.94159958.928286.0567
10002.23283.402810034.77 291.62610056.46290.218610099.84309.710110110.68311.2624
10176.15314.295310214.77307.844110252.94305.869810451.31 309.95210572.61329.4833
10638.78 346.26310704.49351.559810835.41347.866210868.01350.980110965.58350.3716
10987.11358.978910998.95359.7789 11223.4 358.25411340.38398.7141 11533.8411.3204
#Mann= 3 , 0 , 0
9017.764   0.075       09017.764   0.075       0 11533.8   0.075       0
#XS Ineff= 2 , 0
       09797.068        10122.13       0
Bank Sta=9017.764,11533.8
Exp/Cntr=0.3,0.1

Type RM Length L Ch R = 1 ,31252.01,248.843500,248.843500,248.843500
XS GIS Cut Line= 6
 788107.05751879 788555.36335338788483.665209059788426.228985442
789101.097933236788182.640905653789422.907186842 788044.72791446
790002.729030049787782.949131541790524.001146865787566.337357638
#Sta/Elev= 30
8988.112316.67789260.174 318.0189302.683316.66319355.818307.7825 9484.16 311.034
9527.026305.59089720.453307.54239763.521301.74859817.357300.41279828.124 301.294
9838.891307.81189849.658307.13659881.959292.31179946.561293.61369989.759283.2887
10075.92290.436610119.24309.584810148.12311.041910173.38304.674610227.72 303.174
 10512.3303.078710622.13329.1984 10644.1329.186310677.05341.533311049.69346.9267
11093.16355.299411256.17  354.5911321.37386.627311483.45 395.08811600.87396.6009
#Mann= 3 , 0 , 0
8988.112  0.0692       08988.112  0.0692       011600.87  0.0692       0
#XS Ineff= 2 , 0
       09835.288         10138.5       0
Bank Sta=8988.112,11600.87
Exp/Cntr=0.3,0.1

Type RM Length L Ch R = 1 ,31003.17,248.843600,248.843600,248.843600
XS GIS Cut Line= 6
788172.906893317788789.022424274788403.791127618788715.558478728
788627.224805728788638.198015938789043.733616041788476.565281291
789516.684436052788268.261036751790662.687027515787743.614092044
#Sta/Elev= 30
 8957.83315.57879275.476314.26399296.641311.76839317.806302.1546 9423.63300.6784
9820.038301.23519852.389308.8225 9906.51288.09159938.141292.79139971.783284.5069
10004.44283.288410048.12290.893310080.88289.386610135.62309.595410201.29301.3308
10299.81308.042110376.44301.617910552.52305.317310662.66341.860610993.09346.5087
11026.13352.596411059.17349.854511092.21340.375611191.34341.642811257.41356.6214
11312.23375.0041 11323.2370.034311378.02379.599211619.25384.608411660.57392.5804
#Mann= 3 , 0 , 0
 8957.83  0.0634       0 8957.83  0.0634       011660.57  0.0634       0
#XS Ineff= 2 , 0
       09856.039        10141.75       0
Bank Sta=8957.83,11660.57
Exp/Cntr=0.3,0.1

Type RM Length L Ch R = 1 ,30754.33,248.843600,248.843600,248.843600
XS GIS Cut Line= 6
788311.573210161788991.693476339788811.156790173788828.558847877
789059.931143368788736.388013756 789270.20678498788650.347056328
789785.384860856788421.755616739790806.793331714 787927.81954177
#Sta/Elev= 30
9003.711309.67249237.908311.37559279.926310.45579311.603303.31399396.077303.4464
9417.195298.15889778.622300.54199810.869295.31249854.064306.99779897.259 289.128
9951.253292.3499 9972.85283.885410009.87283.307210048.85290.050510081.58288.6282
10125.23308.450210234.35299.961210321.64302.329810384.33312.203510453.18303.5447
10552.05303.130110629.22306.902510651.33314.0121 10684.5315.591510739.78344.1103
11317.53358.241111417.65362.768211462.15379.1603 11528.9 377.31211720.01384.9236
#Mann= 3 , 0 , 0
9003.711  0.0648       09003.711  0.0648       011720.01  0.0648       0
#XS Ineff= 2 , 0
       09853.398        10138.94       0
Bank Sta=9003.711,11720.01
Exp/Cntr=0.3,0.1

Type RM Length L Ch R = 1 ,30505.48,248.843500,248.843500,248.843500
XS GIS Cut Line= 6
788263.786449187  789238.9381207788856.525003457789057.067734197
789381.067894956788876.195030019789553.299347423788809.243806027
790056.954097537788582.212745578790953.833280947788117.585785688
#Sta/Elev= 30
8866.629336.8202 8984.63334.63919024.513311.07959055.837302.25129160.248 308.821
9275.126307.20079306.617301.14579401.087303.60469427.672296.08279696.014302.4379
9738.367287.29979759.558  286.619812.534289.77719854.915306.19579907.892287.9185
10024.48283.187710088.66289.186510131.58 307.19210336.62296.201410440.56303.8922
10513.73293.370310643.86294.100410754.52303.363310795.09 310.27510821.34321.4637
 10955.3323.652211055.94349.526611518.25338.156911603.25379.171511789.02384.8552
#Mann= 3 , 0 , 0
8866.629  0.0684       08866.629  0.0684       011789.02  0.0684       0
#XS Ineff= 2 , 0
       09858.494        10144.23       0
Bank Sta=8866.629,11789.02
Exp/Cntr=0.3,0.1

Type RM Length L Ch R = 1 ,30256.64,248.843600,248.843600,248.843600
XS GIS Cut Line= 6
 788419.65345544789423.144582625789275.731025285789163.377906498
789494.852207043789106.295108392789736.830098989789017.024067442
790462.843007608788660.594860081 791095.75321379788302.367443218
#Sta/Elev= 30
8951.635342.89819017.946340.09349061.162310.66039081.955 302.3169217.113305.9289
9331.942295.91289352.823303.56519405.044304.27529446.998291.62149635.792290.9675
9675.192286.25029814.097289.54349845.563303.64899866.349305.87039914.086286.4224
10072.95280.587410146.48304.629610199.54296.686910307.23291.712710667.62290.5178
10871.64302.763710913.95319.867311097.17318.248911255.84321.500811297.56332.5058
11623.07 334.38311644.34337.931911680.67367.418311715.47381.944911867.16389.4759
#Mann= 3 , 0 , 0
8951.635  0.0701       08951.635  0.0701       011867.16  0.0701       0
#XS Ineff= 2 , 0
       09872.585        10162.15       0
Bank Sta=8951.635,11867.16
Exp/Cntr=0.3,0.1

Type RM Length L Ch R = 1 , 30007.8,248.843500,248.843500,248.843500
XS GIS Cut Line= 6
788784.668217217789624.088426907789224.389508569789484.768093568
789497.949669039789360.564916167790407.996464675788896.386434646
790821.230466275788663.959304917791196.757832723788433.876812836
#Sta/Elev= 30
9238.955301.78469332.602299.53399395.085305.91089520.692307.39789552.359312.4364
9637.147314.00329658.464312.79649726.471293.0105 9765.84287.24449931.048288.3336
9964.382286.63539990.853276.575910042.59281.885810110.36281.213110132.95286.1636
10155.55301.547610166.84303.749810228.97297.456210290.91301.513210316.69 295.293
10380.34290.517810816.34 290.66210906.37 299.04411019.26 301.82511064.81319.2159
11354.36 319.97311394.46 332.28511707.16333.824111805.13383.1435 11937.2389.2211
#Mann= 3 , 0 , 0
9238.955  0.0483       09238.955  0.0483       0 11937.2  0.0483       0
#XS Ineff= 2 , 0
       09858.567        10188.82       0
Bank Sta=9238.955,11937.2
Exp/Cntr=0.3,0.1

Type RM Length L Ch R = 1 ,29758.95,248.843600,248.843600,248.843600
XS GIS Cut Line= 6
788874.159816529789836.441374424 789299.76236999789716.445401202
789543.959567655789613.729813834790567.379510462789083.122458202
790979.168409063788835.628049485791327.016309346788603.475097838
#Sta/Elev= 30
9175.925300.65249259.247298.64719414.375 315.3139560.663313.27639613.293320.5893
9698.759322.76939709.452320.88389785.272284.55519829.107282.18719862.366288.1637
9998.016 274.81410043.48279.862410066.22296.118110077.59299.287710336.68288.1566
10582.23287.911510694.09298.231910842.19290.940110926.71296.499711011.23296.6791
11033.63303.723511068.24308.061911092.48318.359311252.22315.247211381.89318.1124
11429.17333.099511771.78335.129911843.14371.855711860.98384.201511935.05388.3789
#Mann= 3 , 0 , 0
9175.925   0.059       09175.925   0.059       011935.05   0.059       0
#XS Ineff= 2 , 0
       09691.279        10115.44       0
Bank Sta=9175.925,11935.05
Exp/Cntr=0.3,0.1

Type RM Length L Ch R = 1 ,29510.11,248.843600,248.843600,248.843600
XS GIS Cut Line= 6
788937.836811651789987.539328948789296.421948228789910.519787879
789819.798717103789765.824962277790377.365959526789548.003050482
790852.599045513789285.415613207791495.082091891788822.299002632
#Sta/Elev= 30
9196.247302.31659285.111300.9383  9336.2 313.7759458.948316.11139530.791311.7609
  9582.2291.21089667.435282.98139903.128282.860210017.56273.383710038.44279.6689
10048.89291.242610059.33295.330810164.15287.271310351.71288.997310527.49283.2359
10582.95288.522910802.49284.086711064.11290.674511275.22286.677311467.78290.7765
11500.77296.513211552.49318.425911603.94320.082811655.38330.538511889.24334.8486
 11921.6357.098811952.24366.279311977.44380.579912002.64384.336312040.75405.2218
#Mann= 3 , 0 , 0
9196.247  0.0623       09196.247  0.0623       012040.75  0.0623       0
#XS Ineff= 2 , 0
       0                10091.08       0
Bank Sta=9196.247,12040.75
Exp/Cntr=0.3,0.1

Type RM Length L Ch R = 1 ,29261.26,248.843500,248.843500,248.843500
XS GIS Cut Line= 6
789012.216728669790164.034047291789704.282511761790056.790599992
790253.709384645789899.292625575790526.850234472789788.877669144
791038.497455614789477.391781235791626.861284466788993.877280215
#Sta/Elev= 30
9211.529304.40959335.458297.92369446.484313.12349476.764301.46549507.044301.3147
9537.324285.10759567.604 279.676 9587.79 287.5569628.163288.26399668.537280.8223
9882.121280.076910016.23272.010510057.77292.336310390.68277.627210570.27279.9285
10602.37289.811910981.15293.462111060.14 282.99411288.19281.367511348.15287.7764
11639.87281.500211730.35287.793811784.93302.893411808.29315.873911831.94316.7547
11862.64331.690912000.57332.4681 12032.2342.449912107.86350.055612140.23359.1649
#Mann= 3 , 0 , 0
9211.529  0.0528       09211.529  0.0528       012140.23  0.0528       0
#XS Ineff= 2 , 0
       0                10070.58       0
Bank Sta=9211.529,12140.23
Exp/Cntr=0.3,0.1

Type RM Length L Ch R = 1 ,29012.42,393.225100,393.225100,393.225100
XS GIS Cut Line= 6
789072.778075606790307.738938287789987.659323484790269.536615103
 790312.16345048790218.417779177790524.463419706 790147.51590693
790732.990048975790041.888025776791141.005240619789712.600045472
#Sta/Elev= 30
 9238.93305.88389301.338306.49549361.507   300.19391.544311.01149421.582310.3547
9441.607300.02529461.632294.79869521.683291.61919541.689 282.1669561.695  277.95
9601.706280.89469611.709277.93719701.735278.7404 9751.75274.71669791.762280.2254
9991.824271.980910092.01284.412910182.29279.925110282.88288.523410323.35 282.781
10455.74281.920110643.76274.584910807.43276.935610853.51290.400411064.95288.0097
11169.81293.7056 11261.9290.785511314.41294.655611416.72291.556111466.72294.3564
#Mann= 3 , 0 , 0
 9238.93  0.0506       0 9238.93  0.0506       011466.72  0.0506       0
#XS Ineff= 2 , 0
       0                10082.52       0
Bank Sta=9238.93,11466.72
Exp/Cntr=0.3,0.1

Type RM Length L Ch R = 1 , 28619.2,602.149200,602.149200,602.149200
XS GIS Cut Line= 6
789176.362996876 790553.53366676790022.701934457790727.948934019
790278.102339506790699.193814129790793.381247222 790385.33786872
791052.079095393790131.410229012791181.860016197789925.044878215
#Sta/Elev= 30
9384.981308.92089483.698308.0634 9523.82 290.9019604.328286.7579 9624.49277.2741
9644.653273.06519705.621272.03349839.431277.801910008.01269.143510029.18278.7793
10143.96 277.88210185.01281.305110245.62275.7273 10255.7276.169510275.72284.2123
10325.76276.418210426.44271.167210551.03278.741210703.06273.977510941.76 277.234
11011.01 267.55211073.51 267.55211135.38277.778211189.58276.043211233.53279.0388
11252.75284.977411380.32286.471911428.68283.367911463.44 287.57411726.05289.9942
#Mann= 3 , 0 , 0
9384.981  0.0454       09384.981  0.0454       011726.05  0.0454       0
#XS Ineff= 2 , 0
       0                10282.82       0
Bank Sta=9384.981,11726.05
Exp/Cntr=0.3,0.1

Type RM Length L Ch R = 1 ,28017.05,995.374200,995.374200,995.374200
XS GIS Cut Line= 6
789504.588215292791294.063164651790036.780001789791061.308789313
790465.455826938 790809.82799007790848.369612187790482.892944753
791103.518122643790206.231569499791218.629314154 790055.78015992
#Sta/Elev= 30
9859.098316.82799891.921316.05629945.887305.03989978.266267.61179989.502265.6912
 10119.7274.556810163.43 271.63810207.17  275.5810239.97273.557310316.51276.2127
10382.76 272.71610618.76273.452610664.59 278.90310734.44273.235810805.19278.0312
10852.36 273.18810924.91272.018810996.64277.575411062.74273.811211230.56  276.71
11367.12271.639611381.43267.552911466.57 267.55211480.06267.897311508.87276.5576
11577.36275.799711625.71282.968111779.65282.454211837.01 288.35412007.55285.7664
#Mann= 3 , 0 , 0
9859.098  0.0566       09859.098  0.0566       012007.55  0.0566       0
#XS Ineff= 2 , 0
       0                10645.39       0
Bank Sta=9859.098,12007.55
Exp/Cntr=0.3,0.1

Type RM Length L Ch R = 1 ,27021.67,995.374300,995.374300,995.374300
XS GIS Cut Line= 6
789889.743727516792279.371543402790454.486882811791756.498762484
790650.423524825791542.972576149790754.819242538791360.683870013
791049.710393088790653.356797401791330.936285908790188.374256469
#Sta/Elev= 30
9213.658320.41179288.196313.46429315.335303.73219356.045298.49559543.446291.6018
9714.424295.14789731.582280.00929769.417270.17849863.325270.96959910.617265.1649
9955.621 266.7139970.648261.659910012.12261.578110068.29 273.59610245.85272.3824
10271.06266.655110331.33 264.96810377.66277.377310577.11268.074810640.33 269.251
10668.37265.255411182.02272.836611339.64 267.55211362.33273.600111489.32280.6062
11524.56277.201811536.32 283.27611657.28282.988311712.03290.239411794.49291.4164
#Mann= 3 , 0 , 0
9213.658  0.0443       09213.658  0.0443       011794.49  0.0443       0
#XS Ineff= 2 , 0
       0                10255.16       0
Bank Sta=9213.658,11794.49
Exp/Cntr=0.3,0.1

Type RM Length L Ch R = 1 , 26026.3,1446.568100,1446.568100,1446.568100
XS GIS Cut Line= 6
790734.501933429793291.182470893790984.528304884792978.695562415
791099.118761171792717.675567376791073.740403746791160.158928413
791178.073355075790719.210006999791417.241109263790230.397481399
#Sta/Elev= 30
 9046.89288.02139215.614288.08159244.753280.61619325.224277.75799415.941280.3407
9938.301275.31229958.417271.4186 9988.59255.791310008.73253.262210169.56265.7295
10219.56261.987110249.57266.859710369.64263.545510489.94266.637310550.18269.6649
10580.31278.227610650.59280.910510740.88277.742210841.07280.672510861.09276.6154
10921.11276.227310941.11268.600310971.12274.284711151.23270.211711171.28265.2599
11515.38272.582711961.07 267.55212027.82272.5399 12050.2 283.63412295.84288.0599
#Mann= 3 , 0 , 0
 9046.89  0.0453       0 9046.89  0.0453       012295.84  0.0453       0
#XS Ineff= 2 , 0
       09908.794        10817.06       0
Bank Sta=9046.89,12295.84
Exp/Cntr=0.3,0.1

Type RM Length L Ch R = 1 ,24579.73,1041.867500,1041.867500,1041.867500
XS GIS Cut Line= 3
790834.181061864793410.587782875 791961.00215745791944.508723035
792445.656392068791411.389064938
#Sta/Elev= 30
7880.168279.67417925.052280.34987950.277285.64948029.199287.45268063.789 286.093
8094.838277.27548164.689 274.6368265.589276.63768366.488272.08378472.262274.7344
 8587.13271.70788669.187274.59068770.086 270.5748870.986273.2189 8997.11 270.638
9085.398272.78129186.297269.63299779.793269.94069877.249263.70019917.793250.4161
9971.851250.3585 9998.88246.111710025.91246.405710039.42250.084610079.97265.1051
10106.85278.095110121.71289.039810215.11295.360910374.44 329.18610449.74340.2336
#Mann= 3 , 0 , 0
7880.168  0.0642       07880.168  0.0642       010449.74  0.0642       0
#XS Ineff= 2 , 0
       09764.942                       0
Bank Sta=7880.168,10449.74
Exp/Cntr=0.3,0.1

Type RM Length L Ch R = 1 ,23537.86,497.687100,497.687100,497.687100
XS GIS Cut Line= 6
790883.152760838793554.014368636791546.222287945792919.081907613
791742.756418049792783.741411918791949.062419556792734.824362759
792535.152474115792717.056984033 792739.69296994792661.749602517
#Sta/Elev= 30
8442.004279.34228593.855276.86158676.011279.43728705.564272.96118778.759270.3033
8882.191271.75648979.702267.71129078.015270.01579222.152265.97969351.601268.3631
9532.139265.75729634.547267.70179878.831266.31889918.854258.90819958.855239.8773
9968.855 241.0569988.856237.503810018.86237.613810048.86247.398110088.86247.9569
10118.86252.843510148.86270.649110158.87 273.586 10339.1 275.63210419.88279.2908
10430.06 284.17410460.61308.993510470.79314.406810574.84345.2722 10612.1350.7313
#Mann= 3 , 0 , 0
8442.004  0.0451       08442.004  0.0451       0 10612.1  0.0451       0
#XS Ineff= 2 , 0
       0                               0
Bank Sta=8442.004,10612.1
Exp/Cntr=0.3,0.1

Type RM Length L Ch R = 1 ,23040.18,1058.372700,1058.372700,1058.372700
XS GIS Cut Line= 6
790981.278329518793727.511750945791574.913324436793321.402314505
791933.680457044793228.380517133792507.532979973793209.500856662
792660.215238431793140.866926862792813.874595574792978.534981262
#Sta/Elev= 30
8694.383267.89168854.298265.16639042.909266.95429116.088264.48589234.968266.9137
9349.271263.53159448.285265.87049585.774262.76419668.052265.10829769.255262.8326
9879.592264.42139909.596258.6859  9939.6242.27839949.613239.5096 10009.7236.6661
10029.74 237.799 10059.8245.770110069.81246.712610129.82248.109910199.85253.4754
10371.58252.9389 10487.2255.2603 10538.4258.445810551.28260.368110604.46274.6999
10631.26286.504910671.56308.581510697.82318.535210725.43323.466510756.63323.6291
#Mann= 3 , 0 , 0
8694.383  0.0677       08694.383  0.0677       010756.63  0.0677       0
#XS Ineff= 2 , 0
       0                               0
Bank Sta=8694.383,10756.63
Exp/Cntr=0.3,0.1

Type RM Length L Ch R = 1 , 21981.8,932.375800,932.375800,932.375800
XS GIS Cut Line= 6
792341.056686114794776.202629724 792443.12459018794338.742624502
792449.753262656794163.912397806792416.154674991793945.005161056
792434.604189269793847.461558255792881.861500362792976.190355092
#Sta/Elev= 30
9269.775291.42749344.516291.99619396.775289.68159479.448294.81319581.901289.4186
9683.283293.22869713.528284.97999753.704285.20419773.778282.28129903.908285.7215
9913.957280.23569934.054262.84559954.151239.61929974.386230.23639994.762228.7642
10157.01243.723310392.71251.373510527.19 252.48610549.73250.332910651.48249.2803
10742.15252.975610878.16252.504810912.16 256.08210968.94274.2762   11026308.4318
11048.83319.199311071.65326.380111105.89327.988911140.17326.086111196.66307.1012
#Mann= 3 , 0 , 0
9269.775  0.0652       09269.775  0.0652       011196.66  0.0652       0
#XS Ineff= 2 , 0
       0                               0
Bank Sta=9269.775,11196.66
Exp/Cntr=0.3,0.1

Type RM Length L Ch R = 1 ,21049.43,497.687200,497.687200,497.687200
XS GIS Cut Line= 6
793511.067343835794623.206473642793525.760200106794222.593489517
793465.227782084793938.134276849793359.110553997793728.933524222
793074.269407986793374.979652258792974.453670277793171.948164924
#Sta/Elev= 30
8822.689288.2806 8871.28291.20968911.575286.29328961.739288.2874 8992.27285.1824
 9091.89 289.4619262.284287.1492 9404.52290.89769435.528284.01149530.137280.6815
9651.099282.93859685.461266.5812 9697.18  265.059826.898261.90549842.692252.5151
9868.427229.83779874.781227.0255 9912.13229.97099967.519 227.39210026.38229.1305
10092.48235.307810130.92244.6618 10181.1250.2821 10205.8257.401710265.14280.7785
10279.47288.3801 10310.9311.442610322.25316.2127 10377.1324.346510433.12323.9789
#Mann= 3 , 0 , 0
8822.689  0.0512       08822.689  0.0512       010433.12  0.0512       0
#XS Ineff= 2 , 0
       0                               0
Bank Sta=8822.689,10433.12
Exp/Cntr=0.3,0.1

Type RM Length L Ch R = 1 ,20551.74,497.687100,497.687100,497.687100
XS GIS Cut Line= 6
793610.666822723794600.221978514793677.430244179 794009.52020941
793664.801845178793687.607041197793602.511751059793283.939807162
793601.757824759792992.834814684793636.869041792792734.101814108
#Sta/Elev= 30
 8642.26283.29389031.858283.9435 9142.07288.27859162.086284.18079262.145279.8863
9382.166282.14399402.185269.32719422.204264.01349502.368260.75589612.949263.4044
9643.195258.03549764.775256.08319774.939 254.9749825.759230.57399866.415224.1218
9896.907 223.2949947.374227.925410017.52221.085710027.53221.577810067.54 263.409
10077.54 267.61910107.55 253.18510137.56254.070810177.58272.600410257.59301.3883
10337.77337.804110428.56364.357710489.62396.8752 10499.8399.409710521.26413.9755
#Mann= 3 , 0 , 0
 8642.26  0.0515       0 8642.26  0.0515       010521.26  0.0515       0
#XS Ineff= 2 , 0
       0                               0
Bank Sta=8642.26,10521.26
Exp/Cntr=0.3,0.1

Type RM Length L Ch R = 1 ,20054.05,497.687100,497.687100,497.687100
XS GIS Cut Line= 6
793659.534961344794588.944715756 793791.80514467793942.793688124
793885.818627453793674.983387209793969.440766052793538.744138849
794216.295033108793239.348677357794452.313137635792904.409710831
#Sta/Elev= 30
8755.025281.33728994.683284.35339086.296282.44979167.729285.85159281.321283.9474
9320.418279.22949426.999281.37249443.453276.03929453.807268.47339474.515263.7204
9547.651260.31679643.909263.29679677.053256.24829827.638252.1916 9851.09244.3992
9868.246242.53029889.094230.2396   10001216.860510020.68217.294210038.23  221.24
10073.95219.728310100.14230.2747 10126.1236.9504   10133240.796910202.28300.1135
10227.61315.7741 10339.8370.712310467.99419.545710537.59439.179910657.22450.1838
#Mann= 3 , 0 , 0
8755.025  0.0655       08755.025  0.0655       010657.22  0.0655       0
#XS Ineff= 2 , 0
       0                               0
Bank Sta=8755.025,10657.22
Exp/Cntr=0.3,0.1

Type RM Length L Ch R = 1 ,19556.37,497.687100,497.687100,497.687100
XS GIS Cut Line= 6
793991.651711973794381.637899292794059.434177289794261.194174194
794137.108178219794138.370249329794248.803518588793983.178967528
794428.385715216793754.989479767794940.288227234793139.131905809
#Sta/Elev= 30
9276.381278.79339318.249276.98799443.716  279.279457.418276.42919481.135264.9451
9492.914261.73399552.073261.34989588.332 258.3179686.718260.68789727.916252.4019
9809.716249.0943 9876.03250.08449906.801237.85439939.163232.46169971.524216.3934
9990.509214.699810114.89221.9989 10161.7228.937610237.03233.353510328.89233.5706
10407.62229.945310460.01234.2687 10512.1248.489110655.01310.816310680.78324.5625
10722.16341.062710745.19  347.3610770.96350.602510809.47345.4953 10842.4336.3051
#Mann= 3 , 0 , 0
9276.381  0.0503       09276.381  0.0503       0 10842.4  0.0503       0
#XS Ineff= 2 , 0
       0                               0
Bank Sta=9276.381,10842.4
Exp/Cntr=0.3,0.1

Type RM Length L Ch R = 1 ,19058.68,497.687200,497.687200,497.687200
XS GIS Cut Line= 6
794181.117262872 794721.97416663794345.435563948794535.786801164
794456.415819849794420.713386755795042.800501656793841.470823481
795212.052102543793661.280901971795404.679987347793438.262143035
#Sta/Elev= 30
9107.752271.78779206.674269.58349289.525272.20259330.127257.7917 9385.01257.9606
 9482.26254.06499524.071255.53499542.314251.05069627.268247.55919750.077249.1858
9783.017231.75489820.952221.20889853.265223.95269895.353222.24419950.047214.4112
10005.79212.344110022.71 214.71510037.18226.135110047.28228.749710130.42  227.74
10244.02 230.55810621.99229.782710649.52237.431110689.71264.376610703.37271.3347
10729.46273.9016 10755.8280.0665 10819.9289.677710847.82290.844410882.24288.0319
#Mann= 3 , 0 , 0
9107.752  0.0444       09107.752  0.0444       010882.24  0.0444       0
#XS Ineff= 2 , 0
       0                               0
Bank Sta=9107.752,10882.24
Exp/Cntr=0.3,0.1

Type RM Length L Ch R = 1 ,18560.99,497.687100,497.687100,497.687100
XS GIS Cut Line= 6
794333.561939007794995.809973748794665.243486375794730.371217507
795206.928745984794419.416581735795450.714094365794247.108371446
795637.573045618794062.789271268795855.377071747793781.629853753
#Sta/Elev= 30
 9090.78266.13929278.102263.44459303.813259.39849380.304254.32459490.658255.6783
9515.715248.67299563.373248.32229599.111245.10489714.305247.77129726.362243.4156
9762.429223.43079773.892219.89199879.226218.62059910.517  220.199933.182219.0152
 9967.18212.60869989.845211.616610023.91212.374710058.11224.367410458.93225.0032
10526.07227.550610546.83225.026710645.34225.567310668.88223.620910790.66222.7582
10930.69226.564910955.16229.547310972.23234.159411017.06253.762911058.23254.8862
#Mann= 3 , 0 , 0
 9090.78  0.0426       0 9090.78  0.0426       011058.23  0.0426       0
#XS Ineff= 2 , 0
       0                               0
Bank Sta=9090.78,11058.23
Exp/Cntr=0.3,0.1

Type RM Length L Ch R = 1 , 18063.3,497.687100,497.687100,497.687100
XS GIS Cut Line= 6
794563.075380375795408.084118408794943.574497514795129.145581361
795446.397274522794858.333375718795649.986186626794682.463538221
 795839.39906545794416.725325968796487.710489808793262.034379217
#Sta/Elev= 30
9126.518252.41929257.122 256.7939422.443255.87799528.567250.10379740.643251.3128
9752.169249.84549803.065227.88019832.063224.8454 9854.57 217.8469987.623211.1266
 10031.9211.439510065.15218.394810133.37220.460210193.68216.956510449.75223.0531
10963.18219.195411132.84221.9957 11200.7247.341811257.26252.3665 11349.5249.1059
11404.41 231.02311433.81216.821411454.57215.1591 11495.7 223.25711575.58231.4083
11713.96235.2732 11779.6248.530311829.78240.041912005.36249.040712091.53260.2595
#Mann= 3 , 0 , 0
9126.518  0.0426       09126.518  0.0426       012091.53  0.0426       0
#XS Ineff= 2 , 0
       0                11277.87       0
Bank Sta=9126.518,12091.53
Exp/Cntr=0.3,0.1

Type RM Length L Ch R = 1 ,17565.62,497.687100,497.687100,497.687100
XS GIS Cut Line= 6
795040.534414071795978.673368071795371.111489671795664.969553267
795626.313859768795300.043963894795823.939130489794857.369896397
796131.770872161794069.038281609796538.663684862793316.627088207
#Sta/Elev= 30
9096.501241.91169148.249227.95089288.656227.85799328.403223.18219414.437222.0654
9694.927223.82669838.998220.65139857.338214.51339993.312211.118810214.99218.2008
10389.17212.465810454.08218.520910614.89221.3561 11236.7219.468111269.43222.6134
11323.97244.531411345.94248.643811401.03246.918611478.86213.904211523.42221.6888
11612.78221.279411635.42 217.68611669.38228.328411783.78231.069511862.93244.4567
11920.51238.666911989.62240.6755 12035.9249.935212164.92262.219412186.47261.5394
#Mann= 3 , 0 , 0
9096.501  0.0465       09096.501  0.0465       012186.47  0.0465       0
#XS Ineff= 2 , 0
       09737.796           11371       0
Bank Sta=9096.501,12186.47
Exp/Cntr=0.3,0.1

Type RM Length L Ch R = 1 ,17067.93,1493.061400,1493.061400,1493.061400
XS GIS Cut Line= 6
795472.323428711796206.887486839795885.538135843795863.622276978
796097.132680231795453.258506728796132.444000358794411.474075467
796281.631549693793975.104385834796596.257078163793378.334295319
#Sta/Elev= 30
8996.258239.43569246.708239.72899272.341226.7005 9310.79 224.0589690.885224.6546
9747.264219.47689802.484221.41149867.762209.072410018.32206.742610263.09214.3483
10505.21208.252810565.64216.137210675.89219.642511278.21219.616511310.07224.4077
11335.84238.656911352.61242.523611395.54235.940911460.26213.130211536.43225.8904
11657.61223.844111713.17 227.81811746.78220.673711757.98227.080611802.83230.1496
11848.13239.462911870.78237.962111893.43 226.93311904.76 226.53412189.52263.0475
#Mann= 3 , 0 , 0
8996.258  0.0427       08996.258  0.0427       012189.52  0.0427       0
#XS Ineff= 2 , 0
       09650.966         11370.2       0
Bank Sta=8996.258,12189.52
Exp/Cntr=0.3,0.1
